--- PRKRCK.prj (project) ---

Proj Title=PRKRCK
Current Plan=p01
Default Exp/Contr=0,0
English Units
Geom File=g01
Flow File=f01
Plan File=p01
BEGIN DESCRIPTION:
END DESCRIPTION:
DSS Export Rating Curves= 0
DSS Export Rating Curve Sorted= 0
DSS Export Volume Flow Curves= 0
DXF OffsetX= 0
DXF OffsetY= 0
DXF ScaleX= 0
DXF ScaleY= 0

--- PRKRCK.p01 (plan) ---

Plan Title=Floodplain
Program Version=4.00
Geom File=g01
Flow File=f01
K Sum by GR=0
Std Step Tol=0.01
Critical Tol=0.01
Num of Std Step Trials=20
Max Error Tol=0.3
Flow Tol Ratio=0.001
Split Flow NTrial=30
Split Flow Tol=0.02
Split Flow Ratio=0.02
Log Output Level=0
Friction Slope Method=1
Unsteady Friction Slope Method=2
Unsteady Bridges Friction Slope Method=1
Global Log Level=0
CheckData=False
Run HTab=0
Run UNet=0
Run PostProcess=0
UNET Theta=0
UNET Theta Warmup=0
UNET ZTol=0
UNET ZSATol=0
UNET MxIter=0
UNET MaxInSteps=0
UNET DtIC=0
UNET DtMin=0
UNET MaxCRTS=0
UNET WFStab=0
UNET SFStab=0
UNET WFX=0
UNET SFX=0
UNET DSS MLevel=0
UNET DZMax Abort=0
UNET Convert EG Bridges=0
UNET Use Existing IB Tables=0
UNET Froude Limit=0
UNET Froude Power=0
Write IC File=0
Echo Input=False
Echo Output=False
Write Detailed=0

--- PRKRCK.f01 (steady flow) ---

Flow Title=2010 USGS WV Regression Equation
Program Version=4.00
Number of Profiles=1
Profile Names=P100yr
River Rch & RM=PRKRCK,Main      ,15006.9
685.7028
River Rch & RM=PRKRCK,Main      ,12885.3
714.7282
River Rch & RM=PRKRCK,Main      ,11546.5
793.6594
River Rch & RM=PRKRCK,Main      ,7061.7
881.0124
River Rch & RM=PRKRCK,Main      ,4533.8
978.7925
River Rch & RM=PRKRCK,Main      ,1847.8
1013.807
River Rch & RM=PRKRCK,Main      ,1698.6
2018.393
River Rch & RM=PRKRCK,Main      ,289.1
2049.687
Boundary for River Rch & Prof#=PRKRCK,Main      ,1
Up Type=0
Dn Type=3
Dn Slope=0.025379

--- PRKRCK.g01 (geometry) ---

Geom Title=LiDAR
Program Version=4.10

River Reach=PRKRCK          ,Main
Reach XY= 30
     1968935.518      238730.048     1968973.094      238393.723
     1968581.853      238087.425     1969003.165      237475.171
     1968898.971      237185.121     1969149.214      237082.564
     1969029.458      236862.385     1969171.501       236467.09
     1969628.381       236494.37     1970524.908      235753.397
     1970490.881      235463.814     1970674.458      235263.223
     1970790.186      234759.647     1971169.353      234723.536
     1971525.031      234058.366     1971470.047       233736.73
     1971710.868      233280.191     1971755.464      232837.425
     1971468.982      232430.048     1971506.853      232129.786
     1970937.408      231572.147     1971061.019      231132.564
       1970992.8      230380.515     1971535.151      230025.272
     1971858.068      229533.953     1972121.089      229398.536
     1972254.332      229048.679     1971976.124      228092.112
     1971771.263      227964.508     1971611.868         227585.

Type RM Length L Ch R = 1 ,15006.9 ,250,251.9,251.4
XS GIS Cut Line= 3
     1969252.461      238422.967     1969179.123      238544.086
     1968779.095      238714.098
#Sta/Elev= 30
       0 2263.14    77.2 2242.61    86.9 2240.99    96.5 2238.79   106.2 2238.56
   109.4 2238.17   119.1 2236.12   128.7 2233.63   148.1  2230.8   157.9  2230.4
   174.3 2229.06     220 2227.73   239.6 2227.57     269    2228   321.3 2226.24
   344.2 2227.07   347.5 2226.87   350.8 2225.98     354 2224.31   357.3 2223.12
   360.6 2223.17   367.1  2224.4   373.6 2225.01   380.2  2226.1   396.5 2226.36
   416.1 2227.55   458.6 2228.33   484.7 2230.24   517.4 2230.21   576.2 2231.36
#Mann= 3 ,-1 , 0
       0     .12       0     354    .045       0   367.1     .12       0
Bank Sta=354,367.1
XS Rating Curve= 0 ,0
Exp/Cntr=0.3,0.1

Type RM Length L Ch R = 1 ,14755.1 ,324.9,318.1,310.9
XS GIS Cut Line= 3
     1969200.721       238341.43     1968796.249      238505.885
     1968676.241       238491.44
#Sta/Elev= 30
       0 2258.67     9.8    2256    32.6 2250.76    61.9 2243.46    68.4 2242.57
      88 2241.43   104.3 2239.68   117.3 2237.58   143.4 2234.19   156.4 2231.86
   198.8 2225.76   215.1 2225.12   221.6 2223.99   228.1 2223.31   232.5 2224.01
   237.9 2225.43   254.2 2226.63   273.7 2226.05   316.1 2226.36   335.6 2225.84
   345.4  2226.4   371.5 2226.87     391 2227.96   423.6 2227.84   459.5 2228.33
   479.1 2229.21   498.7  2230.7   521.6 2233.68   534.6 2234.29   557.5 2236.12
#Mann= 3 ,-1 , 0
       0     .12       0   221.6    .045       0   232.5     .12       0
Bank Sta=221.6,232.5
XS Rating Curve= 0 ,0
Exp/Cntr=0.3,0.1

Type RM Length L Ch R = 1 ,14436.9 ,167.7,165.9,164.1
XS GIS Cut Line= 2
     1968906.233      238176.224     1968647.327      238390.683
#Sta/Elev= 30
       0 2235.07     9.8 2231.66    13.1 2230.72    16.3 2230.24    26.1 2230.53
    52.2 2229.75    58.8 2230.03    65.3 2229.76    71.8 2229.84    75.1 2229.53
    88.1  2229.2    97.9 2229.28     111 2228.48   140.4 2227.19   166.5 2226.74
   169.7 2226.49     173    2226   182.8 2222.99     186  2222.5   195.8 2221.83
   199.1 2221.81  201.67 2222.54   205.6  2223.6   208.9 2224.09   248.1 2226.94
   254.6 2227.18   274.2 2227.37     284 2228.03   316.6 2230.74   336.2 2231.75
#Mann= 3 ,-1 , 0
       0     .12       0     186    .045       0  201.67     .12       0
#XS Ineff= 2 , 0
          167.23  2227.7
Permanent Ineff=
       F       F
Bank Sta=186,201.67
XS Rating Curve= 0 ,0
Exp/Cntr=0.3,0.1

Type RM Length L Ch R = 1 ,14271   ,209.8,236.6,261.7
XS GIS Cut Line= 3
     1968858.084      238140.173     1968683.564      238146.333
     1968568.586      238259.257
#Sta/Elev= 30
       0 2230.44     6.5 2230.19    32.3 2228.09      42 2227.97    64.7 2226.96
    90.6 2226.75   100.2 2226.28     110 2226.33   122.9 2225.83   135.8 2224.74
   142.3 2224.77   158.5 2225.72   161.7  2225.6   181.1 2223.61   190.7  2223.5
     194 2223.14   200.4 2221.44   206.9 2220.95   216.5 2220.56   222.8 2221.03
   226.2 2221.61   232.6 2223.34   239.1 2224.77   245.5 2225.87   248.8 2226.17
     281 2228.06   293.9 2228.31     310 2229.04   322.9 2229.22   335.8 2230.06
#Mann= 3 ,-1 , 0
       0     .12       0   206.9    .045       0   222.8     .12       0
Bank Sta=206.9,222.8
XS Rating Curve= 0 ,0
Exp/Cntr=0.3,0.1

Type RM Length L Ch R = 1 ,14034.4 ,184.3,187.7,190.7
XS GIS Cut Line= 2
      1968784.17      238051.887     1968502.885      237945.121
#Sta/Elev= 30
       0 2228.75    16.4  2227.2    32.7 2225.15      49 2225.22    65.4 2223.39
    98.1 2222.16     121 2219.36   124.3 2218.65   127.5 2217.31   130.8 2214.76
   134.1 2211.64   137.4 2209.43   139.5 2208.73   143.9 2207.91   147.2 2207.92
   154.5 2208.89   160.2 2210.32   163.5 2211.74   173.3 2217.57   176.6 2219.26
   179.9 2220.46   183.1  2220.9   189.7 2220.94   202.8 2222.18   215.8  2224.1
   235.5 2226.35   251.8 2228.83   268.2 2232.24     278 2234.63   300.9 2241.37
#Mann= 3 ,-1 , 0
       0     .12       0   139.5    .045       0   154.5     .12       0
Bank Sta=139.5,154.5
XS Rating Curve= 0 ,0
Exp/Cntr=0.3,0.1

Type RM Length L Ch R = 1 ,13846.8 ,165.9,168.8,171.6
XS GIS Cut Line= 2
     1968827.286      237887.633     1968589.118      237756.229
#Sta/Elev= 30
       0 2225.41    13.1 2224.98    49.2 2219.67    68.8 2217.76    72.1 2216.95
    75.4 2215.61    85.2 2210.15      95 2204.02    98.3 2202.62   101.6 2201.81
  106.29  2201.2   114.7 2200.56     118 2200.58   121.3 2201.21   124.5 2202.72
   131.1 2206.84   134.4 2209.28   140.9 2214.73   144.2 2216.86   147.5 2218.11
   150.8 2218.73   157.3 2219.18   170.4  2219.4     177 2220.35   206.5 2222.62
   216.3  2224.7   239.2 2231.02   245.8 2232.41   252.4 2234.42     272  2239.4
#Mann= 3 ,-1 , 0
       0     .12       0  106.29    .045       0   121.3     .12       0
Bank Sta=106.29,121.3
XS Rating Curve= 0 ,0
Exp/Cntr=0.3,0.1

Type RM Length L Ch R = 1 ,13678   ,126.9,127.4,127.9
XS GIS Cut Line= 2
     1968890.935       237743.91     1968726.681      237624.826
#Sta/Elev= 30
       0 2209.04     3.3 2208.88    13.1 2209.15    16.4 2208.95      36 2205.95
    39.3 2204.74    42.5 2203.19    49.1 2199.34    55.6    2196    62.2 2193.45
    65.4 2192.73      72 2192.11    75.3 2192.16    78.5 2192.63    81.8 2193.59
    88.4 2196.65    94.9 2200.49   101.4 2204.82   104.7  2206.7   111.3  2209.1
   114.5 2209.93   124.4 2210.74   127.6 2210.76   134.2 2210.27   147.2 2210.18
   157.1 2210.87   173.4 2212.58     180 2213.99   189.8 2217.38   202.9 2222.29
#Mann= 3 ,-1 , 0
       0     .12       0    65.4    .045       0    78.5     .12       0
Bank Sta=65.4,78.5
XS Rating Curve= 0 ,0
Exp/Cntr=0.3,0.1

Type RM Length L Ch R = 1 ,13550.6 ,147.4,147.9,148.3
XS GIS Cut Line= 2
     1968978.483      237652.494     1968830.696      237540.264
#Sta/Elev= 30
       0 2204.41     9.8 2203.97    19.5 2203.34      26  2203.3    35.8 2202.87
    45.6 2202.04    52.1 2201.79    55.4 2200.66    58.6 2199.23    61.9 2197.53
    65.1 2195.44    71.6 2190.68    74.9 2188.85    78.1 2187.93    81.4 2187.44
    91.2 2186.91    94.4 2187.16   95.77  2187.5    97.7 2187.96   107.4 2191.02
   110.7 2192.51     114 2194.49   120.5 2199.17   123.7 2201.05   130.2  2203.3
   143.2 2204.21   162.8 2204.74   175.8 2205.86   182.3 2206.11   185.6 2206.41
#Mann= 3 ,-1 , 0
       0     .12       0    81.4    .045       0   95.77     .12       0
Bank Sta=81.4,95.77
XS Rating Curve= 0 ,0
Exp/Cntr=0.3,0.1

Type RM Length L Ch R = 1 ,13402.7 ,224.3,196,166.4
XS GIS Cut Line= 3
     1969065.156      237534.708     1968959.593      237451.369
     1968868.476      237459.147
#Sta/Elev= 30
       0 2197.87     6.6 2197.57      23 2197.51    32.8  2197.1    36.1 2196.71
    42.6 2195.35    49.2 2193.49    52.5 2191.83    68.9 2182.49    72.2 2180.84
    75.4 2179.78    78.7 2179.46      82 2179.43    88.6  2179.7    98.4 2182.28
     105 2183.07   108.2 2183.99   114.8 2186.62   121.4 2188.27   127.9 2189.48
   144.3 2191.44   157.4 2193.96   167.2 2194.84   183.5 2194.68   196.6 2195.61
   203.1 2195.86   209.6 2196.67   212.9 2197.32   219.4 2198.72   225.9 2200.45
#Mann= 3 ,-1 , 0
       0     .12       0    75.4    .045       0    88.6     .12       0
Bank Sta=75.4,88.6
XS Rating Curve= 0 ,0
Exp/Cntr=0.3,0.1

Type RM Length L Ch R = 1 ,13206.7 ,114.5,144.3,171.7
XS GIS Cut Line= 2
     1969022.251      237262.398     1968870.252      237367.078
#Sta/Elev= 30
       0 2177.04     6.5 2176.36    16.2    2175    29.1 2173.83    42.1 2174.35
    45.3 2173.63    48.6 2172.53    51.8 2170.88      55 2169.64    58.3  2169.4
    64.8 2169.51      68 2169.76    77.7 2172.05    84.2 2173.04    87.4 2173.06
    90.7 2172.81   100.4 2173.12   106.8 2172.79   116.6 2174.35   119.8 2174.58
   126.3 2174.51   129.5 2175.39   132.8 2177.22   139.2 2182.23   142.5 2184.51
   145.7 2186.25   148.9 2187.35   168.4 2190.16   178.1 2192.32   184.6 2193.48
#Mann= 3 ,-1 , 0
       0     .12       0      55    .045       0      68     .12       0
#XS Ineff= 2 , 0
                           85.04         2175.39
Permanent Ineff=
       F       F
Bank Sta=55,68
XS Rating Curve= 0 ,0
Exp/Cntr=0.3,0.1

Type RM Length L Ch R = 1 ,13062.5 ,51.7,66.9,84
XS GIS Cut Line= 3
       1969009.9      237261.884     1968863.372      237155.634
     1968817.539      237168.829
#Sta/Elev= 30
       0 2173.22     9.7  2170.7    19.4 2169.21    38.8 2164.31      42 2163.94
    45.2 2164.22    51.7 2165.93      55 2166.39    64.6 2166.42    71.1 2167.01
    80.8 2167.14    87.3 2167.81    90.5  2167.8   100.2 2165.88   106.7 2165.07
   122.8 2165.27   129.3  2164.1   132.5 2163.62   135.8 2163.52   142.2 2163.91
   145.4 2164.68   148.7 2166.57   161.6 2176.55   164.8 2178.78   174.5 2182.12
   177.8 2183.07   193.7 2184.87   209.6 2187.33   219.2 2189.86   228.7 2192.95
#Mann= 3 ,-1 , 0
       0     .12       0   129.3    .045       0   142.2     .12       0
Bank Sta=129.3,142.2
XS Rating Curve= 0 ,0
Exp/Cntr=0.3,0.1

Type RM Length L Ch R = 1 ,12995.6 ,111.9,110.3,105.8
XS GIS Cut Line= 3
     1969016.497      237256.476     1968966.584      237183.776
     1968945.968       237077.44
#Sta/Elev= 30
       0 2174.19     9.8 2170.48    19.6 2167.31    29.4 2162.92    32.7 2162.24
    39.2 2162.13    55.5 2163.97    58.8 2163.95    65.3 2163.32    75.1 2163.87
    88.2 2162.49    97.7 2160.08   100.9 2159.72   107.3 2159.27   113.7 2159.78
   116.9 2160.67     120 2162.05   123.2 2164.57   129.6 2170.21   132.8 2172.61
     136 2174.64   139.2 2176.35   142.3 2177.49   145.5 2178.07   155.1 2177.61
   164.6 2177.89   174.2 2177.64   183.8 2176.49   193.3 2176.76   196.5 2176.44
#Mann= 3 ,-1 , 0
       0     .12       0   100.9    .045       0   113.7     .12       0
Bank Sta=100.9,113.7
XS Rating Curve= 0 ,0
Exp/Cntr=0.3,0.1

Type RM Length L Ch R = 1 ,12885.3 ,194.3,164.1,133.3
XS GIS Cut Line= 3
      1969106.27      237240.243     1969048.488      237093.567
     1968970.705      237066.898
#Sta/Elev= 30
       0  2182.9    16.1 2181.63    22.5  2180.6    25.7 2179.61      29 2177.79
    35.4 2172.69      45 2166.12    51.5 2160.27    54.7 2157.91    57.9 2156.57
    61.1 2156.11    70.8 2156.29    90.1 2153.63    96.5 2153.15    99.7 2153.57
   106.2 2155.78   122.3 2158.05   128.7 2157.99   135.1 2156.88   141.6 2156.56
   151.2    2158     164 2158.86   167.1  2159.6   170.3 2161.08     183 2168.33
   186.1 2169.74   195.6  2172.6   198.8  2173.1   220.9 2173.98   239.9  2173.7
#Mann= 3 ,-1 , 0
       0     .12       0    90.1    .045       0    99.7     .12       0
#XS Ineff= 2 , 0
           70.95 2158.81   124.1         2159.16
Permanent Ineff=
       F       F
Bank Sta=90.1,99.7
XS Rating Curve= 0 ,0
Exp/Cntr=0.3,0.1

Type RM Length L Ch R = 1 ,12721.2 ,222.7,235.4,246
XS GIS Cut Line= 2
       1969218.5      237019.117     1968964.038      237055.786
#Sta/Elev= 30
       0 2181.87     9.8 2178.49    19.5 2176.64      26  2174.8    29.3 2173.37
    35.8 2168.43    42.3 2162.32    52.1 2150.88    55.3    2149    58.6 2148.19
    61.8 2147.79    71.6 2147.68    76.4 2148.16    81.4 2149.05    94.4 2149.96
   100.9 2149.64   123.7 2149.45   136.7  2148.2   149.7 2149.66   156.2 2151.09
     166  2154.4   175.7 2158.56     179 2160.26   188.8 2166.65     192 2168.13
   198.5 2170.02   208.3 2171.66   234.3 2172.88   244.1 2172.97   257.1 2174.35
#Mann= 3 ,-1 , 0
       0     .12       0    58.6    .045       0    76.4     .12       0
#XS Ineff= 2 , 0
                           96.28         2151.55
Permanent Ineff=
       F       F
Bank Sta=58.6,76.4
XS Rating Curve= 0 ,0
Exp/Cntr=0.3,0.1

Type RM Length L Ch R = 1 ,12485.7 ,198.4,202.3,205.2
XS GIS Cut Line= 3
      1969209.61      236912.443     1968988.484      236832.438
     1968930.702       236862.44
#Sta/Elev= 30
       0 2160.94     9.8 2158.41    16.3 2157.44    42.5 2155.45      49 2153.73
      62 2147.81    68.6  2146.1    94.7 2147.21      98 2146.52   114.3 2140.12
   117.6 2139.19   120.8 2138.86   130.6 2140.16   143.7 2140.09   150.2 2139.44
   156.8 2139.44   169.8 2137.22   182.9 2137.03   189.4 2136.48   192.7 2136.52
  194.07 2137.07     196 2137.85   199.2 2140.28   218.8 2157.66   222.1 2159.95
   225.4 2161.42   261.2 2170.78   277.5 2176.32   287.2    2179   300.3 2184.17
#Mann= 3 ,-1 , 0
       0     .12       0   182.9    .045       0  194.07     .12       0
Bank Sta=182.9,194.07
XS Rating Curve= 0 ,0
Exp/Cntr=0.3,0.1

Type RM Length L Ch R = 1 ,12283.4 ,181.3,169.5,157.2
XS GIS Cut Line= 2
     1969254.058      236759.099      1969040.71      236641.313
#Sta/Elev= 30
       0 2157.14      13 2152.59    16.2 2151.24    22.8 2149.54      52 2140.41
    68.2 2133.18      78  2129.5   86.47 2125.36    87.7 2124.86      91 2124.52
   100.4 2125.34   107.2 2126.76   110.5 2127.08     117 2126.66   123.5 2127.48
   139.7 2132.52   146.2 2135.77   152.7 2138.14   162.5 2140.72   165.7 2141.13
   175.5 2141.71   185.2 2141.25   191.7 2141.27   201.5 2142.14   214.5 2142.56
   217.7 2142.42   224.2 2141.52   227.5 2141.43   237.2 2142.73   243.7 2142.81
#Mann= 3 ,-1 , 0
       0     .12       0   86.47    .045       0   100.4     .12       0
Bank Sta=86.47,100.4
XS Rating Curve= 0 ,0
Exp/Cntr=0.3,0.1

Type RM Length L Ch R = 1 ,12113.9 ,173.9,212.9,248.9
XS GIS Cut Line= 2
     1969267.392      236545.751     1969050.711      236551.307
#Sta/Elev= 30
       0 2121.22    22.6 2123.74    32.4  2123.8    42.1 2124.54    45.3 2124.54
      55 2123.17    61.5  2123.2    67.9 2122.62    71.2 2121.89    74.4 2120.66
    77.6 2119.07    84.1 2116.71   92.02 2115.17      97 2114.84   103.5 2115.17
     110 2116.62   116.5 2118.58   119.7 2119.82   122.9 2121.31   126.2 2123.33
   132.6 2128.39   135.9 2130.44   148.8 2136.57   155.3 2138.75   158.5 2139.44
   168.2 2140.68   177.9 2141.38   197.3 2143.47   203.8 2143.99   216.8 2144.49
#Mann= 3 ,-1 , 0
       0     .12       0   92.02    .045       0   103.5     .12       0
Bank Sta=92.02,103.5
XS Rating Curve= 0 ,0
Exp/Cntr=0.3,0.1

Type RM Length L Ch R = 1 ,11901   ,128.8,124.1,117.4
XS GIS Cut Line= 3
     1969287.393      236534.639     1969289.616      236402.408
      1969265.17      236351.294
#Sta/Elev= 30
       0 2119.71    12.9 2118.54    19.4 2119.01    22.6 2118.94      29 2118.08
    35.5 2116.24    41.9 2112.11    51.6 2108.33    54.8 2107.59    58.1  2107.6
    64.5 2107.36      71 2107.63    80.6 2107.67    96.8 2106.57     100 2107.06
   109.7 2109.29   116.1 2111.24   119.4 2112.56   122.6 2114.14   125.8 2115.89
   132.2 2120.22   135.4 2122.14   144.8 2128.64     148  2131.3   157.4 2140.47
   160.6 2142.84   163.7 2144.45   166.9 2145.49   173.2 2146.76   188.9 2154.58
#Mann= 3 ,-1 , 0
       0     .12       0    58.1    .045       0      71     .12       0
Bank Sta=58.1,71
XS Rating Curve= 0 ,0
Exp/Cntr=0.3,0.1

Type RM Length L Ch R = 1 ,11776.9 ,224.6,230.3,235.1
XS GIS Cut Line= 3
     1969439.132      236583.867     1969390.734      236382.407
     1969384.067      236331.292
#Sta/Elev= 30
       0 2152.53    16.2  2142.3    25.9 2135.52    32.4 2129.43    51.8 2113.14
    58.3  2108.3    61.5 2106.62    71.2 2104.12    84.2 2105.32    97.1 2105.69
   106.8 2106.96   110.1 2106.68   119.8 2104.19   132.7 2104.51     136 2103.64
   142.4 2100.48   148.9 2099.44     154 2100.35   158.6 2101.56   165.1 2102.12
   178.1 2100.58   181.3 2100.64   184.5 2101.71   194.2 2109.92   213.6  2124.1
   223.3 2132.33   226.5 2134.46     233 2137.67   249.1 2143.29   258.7 2148.06
#Mann= 3 ,-1 , 0
       0     .12       0   142.4    .045       0     154     .12       0
Bank Sta=142.4,154
XS Rating Curve= 0 ,0
Exp/Cntr=0.3,0.1

Type RM Length L Ch R = 1 ,11546.5 ,162.7,151.4,139.9
XS GIS Cut Line= 3
     1969601.333      236577.707     1969601.859      236423.521
     1969568.524      236339.071
#Sta/Elev= 30
       0  2160.2    19.7 2147.48    49.2  2130.8    55.8 2126.42      59 2123.47
    62.3 2118.99    65.6 2110.32    68.9 2101.02    72.2 2093.14    75.4 2089.87
    78.7 2088.88      82 2088.92    88.1 2089.79     105 2091.17   108.3 2091.95
   111.5 2093.64   114.8 2094.76   124.7 2094.86   127.9 2095.66   131.2 2097.07
   134.5 2097.66   154.2  2097.9   170.4 2102.99   183.4 2109.82   189.9 2112.51
   199.6 2114.83   212.6 2118.86   225.5 2121.59     232 2123.94     245 2129.47
#Mann= 3 ,-1 , 0
       0     .12       0    75.4    .045       0    88.1     .12       0
Bank Sta=75.4,88.1
XS Rating Curve= 0 ,0
Exp/Cntr=0.3,0.1

Type RM Length L Ch R = 1 ,11395.2 ,148.6,146.1,143.4
XS GIS Cut Line= 2
     1969775.853      236505.846     1969685.198      236337.959
#Sta/Elev= 30
       0 2124.29    25.9  2115.5    29.1 2114.04    32.3 2111.85    38.8  2106.4
    45.3 2101.75    48.5 2098.99    58.2 2089.61    61.4 2087.03    64.7 2085.71
   76.46  2083.2    80.8 2082.97    87.3  2083.2    93.8 2084.26      97 2085.92
   106.7 2089.74     110 2090.34   116.4 2090.42   122.9 2089.76   126.1 2090.14
   132.6 2092.41   135.8 2092.74   145.5 2093.63   148.8 2093.65   155.2 2093.04
   158.5 2094.04   168.2 2098.13   174.6 2101.35   184.3 2105.64   190.8 2107.85
#Mann= 3 ,-1 , 0
       0     .12       0   76.46    .045       0    87.3     .12       0
Bank Sta=76.46,87.3
XS Rating Curve= 0 ,0
Exp/Cntr=0.3,0.1

Type RM Length L Ch R = 1 ,11249   ,157.4,156.1,154.2
XS GIS Cut Line= 3
     1969876.459      236448.357     1969871.878      236373.517
     1969799.651      236270.177
#Sta/Elev= 30
       0 2107.66     6.5 2105.82    16.3 2104.36    26.1 2101.84    39.1 2099.98
    55.4 2096.89    65.2 2094.64      75  2091.5    78.2 2089.39    84.7 2084.07
    87.9  2082.1    91.1 2081.32    97.6 2081.73   104.1 2080.09  113.01 2078.95
   120.2 2078.55   124.7 2078.93   133.2 2079.31   136.4 2080.11   142.9 2083.55
   146.1 2084.19   152.6 2083.42   165.5 2083.88   168.7 2084.59     172 2085.98
   178.4 2089.94   181.7 2092.67   188.1  2099.8   197.8 2109.92   201.1 2113.89
#Mann= 3 ,-1 , 0
       0     .12       0  113.01    .045       0   124.7     .12       0
Bank Sta=113.01,124.7
XS Rating Curve= 0 ,0
Exp/Cntr=0.3,0.1

Type RM Length L Ch R = 1 ,11092.9 ,207.1,197.9,187.3
XS GIS Cut Line= 2
     1970055.085      236353.911     1969919.659      236186.838
#Sta/Elev= 30
       0 2081.81    22.8 2079.15    32.6 2078.67    35.8 2078.78    58.6 2081.44
    71.7    2082      75 2081.85    84.7 2079.88    91.2 2077.76    97.8 2076.63
     101 2075.63   107.5 2072.21  110.07 2071.68     114 2071.44   120.6 2071.63
   127.1 2071.62   136.9 2072.52   140.1 2072.95   146.6  2074.4   153.2 2075.23
   156.4 2076.41   159.7 2079.02   162.9 2082.26   166.2 2086.71     176 2102.43
   179.2 2106.57   195.5  2123.2     202 2129.42   211.8 2137.23   215.1 2139.56
#Mann= 3 ,-1 , 0
       0     .12       0  110.07    .045       0   120.6     .12       0
Bank Sta=110.07,120.6
XS Rating Curve= 0 ,0
Exp/Cntr=0.3,0.1

Type RM Length L Ch R = 1 ,10895.1 ,161.5,169.6,177.7
XS GIS Cut Line= 2
      1970239.87      236187.604     1970010.776      236074.608
#Sta/Elev= 30
       0 2081.85    16.4 2080.32    29.5 2076.59    42.6 2075.38    49.1 2073.17
      59 2068.55    65.5 2066.67      72 2066.51    98.2 2068.87   101.5 2068.73
   114.6 2065.87   117.9 2065.58   127.7 2065.39   134.3 2065.45   150.6 2067.77
   163.8 2065.75     167 2065.82   170.3 2067.27   173.6 2070.47   183.4 2081.99
     190 2087.23   193.2 2090.27   199.8 2097.67   212.9 2110.34   219.4 2118.09
   222.7  2121.2   232.5 2128.49   239.1 2132.71   245.6 2138.12   255.4 2145.08
#Mann= 3 ,-1 , 0
       0     .12       0   117.9    .045       0   134.3     .12       0
#XS Ineff= 2 , 0
           98.45 2072.84
Permanent Ineff=
       F       F
Bank Sta=117.9,134.3
XS Rating Curve= 0 ,0
Exp/Cntr=0.3,0.1

Type RM Length L Ch R = 1 ,10725.5 ,163.5,171.1,177.7
XS GIS Cut Line= 2
     1970287.093       236113.69      1970098.56      235916.819
#Sta/Elev= 30
       0 2077.07    16.2 2070.54    22.7 2067.62      26 2066.59    48.7 2063.13
    61.7 2062.68    71.4 2063.03    81.1  2062.9   103.8 2060.68   116.8  2062.2
   129.8 2062.55   139.5 2061.75   149.3 2061.34   155.8 2061.45     172 2059.72
   178.5 2060.19     185 2059.55   191.5 2059.38     198 2058.32   201.2 2058.16
   204.4 2058.51   207.7 2059.61   210.9 2061.84   217.4 2067.87   236.9 2084.15
   243.4 2091.13   249.9 2099.37   253.1 2102.94   266.1 2115.25   272.6 2120.48
#Mann= 3 ,-1 , 0
       0     .12       0   191.5    .045       0   207.7     .12       0
#XS Ineff= 2 , 0
          126.63 2065.27
Permanent Ineff=
       F       F
Bank Sta=191.5,207.7
XS Rating Curve= 0 ,0
Exp/Cntr=0.3,0.1

Type RM Length L Ch R = 1 ,10554.4 ,161.9,159.4,156.9
XS GIS Cut Line= 2
     1970363.061      236025.403     1970252.189      235797.501
#Sta/Elev= 30
       0 2073.54     6.5 2070.43    16.2 2063.97    22.7 2060.18    32.5 2055.98
      39 2055.35      52 2056.61    68.2 2055.11      78 2056.72   107.2 2057.83
   110.5 2057.57   113.7 2056.29   123.5 2050.38   126.7 2049.05   129.7 2048.58
   133.2 2048.52   146.2 2048.73     156 2052.02   159.2 2052.41     169 2051.81
   172.2 2052.08   185.2 2055.22   214.4 2053.91   224.2 2054.68   227.4 2056.15
   230.7  2058.4   240.4 2066.08   246.9 2070.39   250.2 2072.52   253.4 2073.79
#Mann= 3 ,-1 , 0
       0     .12       0   129.7    .045       0   146.2     .12       0
#XS Ineff= 2 , 0
                          160.06         2053.56
Permanent Ineff=
       F       F
Bank Sta=129.7,146.2
XS Rating Curve= 0 ,0
Exp/Cntr=0.3,0.1

Type RM Length L Ch R = 1 ,10395   ,240.6,222.9,204.9
XS GIS Cut Line= 4
     1970533.474      235891.947     1970456.362      235846.815
     1970383.672      235731.749     1970309.678      235694.842
#Sta/Elev= 30
       0 2119.75    28.7 2101.95    31.9 2099.34    70.2 2055.39    76.6 2049.52
    79.8 2048.09    86.2 2046.73    89.4 2045.61    95.8 2045.09   105.6  2045.5
     112 2043.73   118.6 2043.18   131.5 2042.81   134.7 2043.01     138 2044.01
   141.2 2045.74   144.4  2046.9   147.7 2047.56   176.8  2045.1   186.6 2045.62
   189.8 2046.34     193 2047.63     206  2054.2   209.2 2055.22   212.5 2055.54
   225.4 2055.22   260.4 2057.01   279.5 2061.18   295.4  2067.8   308.1 2074.25
#Mann= 3 ,-1 , 0
       0     .12       0   118.6    .045       0   134.7     .12       0
#XS Ineff= 2 , 0
          104.02 2049.46  148.45         2050.81
Permanent Ineff=
       F       F
Bank Sta=118.6,134.7
XS Rating Curve= 0 ,0
Exp/Cntr=0.3,0.1

Type RM Length L Ch R = 1 ,10172.1 ,220.5,220.3,219
XS GIS Cut Line= 2
     1970687.462      235678.417     1970340.476      235602.449
#Sta/Elev= 30
       0 2122.81      13 2116.02    22.8 2109.95    42.4 2095.89    55.4 2087.15
    65.2 2079.07    71.7 2073.36      75 2068.52    78.2 2062.97    81.5 2059.02
    94.5 2040.08    97.8 2036.66     102 2034.32   107.5 2033.54     117 2034.43
   127.1 2036.99   133.6 2038.02   153.2 2037.63   172.7 2036.13   182.5 2037.52
   195.5 2036.24     202 2036.05   215.1 2036.66   247.7 2036.75   254.2 2037.52
   260.7 2040.57   270.5 2046.59   296.6 2057.41   325.9 2067.78   355.2 2082.32
#Mann= 3 ,-1 , 0
       0     .12       0     102    .045       0     117     .12       0
#XS Ineff= 2 , 0
                           135.4         2041.89
Permanent Ineff=
       F       F
Bank Sta=102,117
XS Rating Curve= 0 ,0
Exp/Cntr=0.3,0.1

Type RM Length L Ch R = 1 ,9951.8  ,155.3,170.7,185.6
XS GIS Cut Line= 2
      1970673.09      235497.737       1970360.8      235439.009
#Sta/Elev= 30
       0 2080.62    16.4 2073.22    42.6 2063.72    52.4 2059.68    72.1 2055.25
      95 2048.97   101.6 2046.14   124.5 2033.72     131 2031.89   137.6 2030.95
   147.4  2031.5   157.2 2030.22   173.6 2024.01   183.4 2023.29   186.7 2023.87
   196.6 2025.78   206.4 2025.76   216.2 2024.85   229.3 2025.46   235.9 2026.64
   242.4 2028.52     249 2031.67   258.8 2039.66   265.4 2046.69   275.2 2055.28
   278.4 2058.82   288.3 2072.38   294.8 2080.17   311.2 2093.12   317.8 2097.37
#Mann= 3 ,-1 , 0
       0     .12       0   173.6    .045       0   186.7     .12       0
#XS Ineff= 2 , 0
                          199.74         2030.54
Permanent Ineff=
       F       F
Bank Sta=173.6,186.7
XS Rating Curve= 0 ,0
Exp/Cntr=0.3,0.1

Type RM Length L Ch R = 1 ,9781.2  ,161.5,150.8,139.9
XS GIS Cut Line= 4
     1970706.864      235402.063     1970639.082      235382.061
     1970552.409      235283.166     1970467.959      235246.496
#Sta/Elev= 30
       0 2082.56    28.9 2066.14    38.6 2061.62    51.4 2054.74    70.7 2046.39
    73.9 2044.33    77.1 2041.28    89.9 2027.71   102.8 2015.18     106 2012.43
   109.2 2010.85   112.4 2009.79   118.8 2009.14   125.2 2009.65   131.6  2010.2
   141.2 2012.52   166.9 2017.49   173.3 2019.58   182.9  2023.6   186.1 2024.13
   195.8 2023.96   208.5 2021.25   211.7 2020.92     218  2021.5   233.9 2026.16
   246.6  2031.4   259.3 2035.39   278.4 2043.59   287.9 2048.33   294.2 2050.06
#Mann= 3 ,-1 , 0
       0     .12       0   112.4    .045       0   125.2     .12       0
Bank Sta=112.4,125.2
XS Rating Curve= 0 ,0
Exp/Cntr=0.3,0.1

Type RM Length L Ch R = 1 ,9630.3  ,170.8,167.8,164.9
XS GIS Cut Line= 2
      1970754.16      235248.996     1970551.924      235168.991
#Sta/Elev= 30
       0 2087.71    16.2 2075.61    29.2 2064.11    35.7 2059.18      39  2056.3
    42.2 2052.03    48.7 2042.63    55.2 2032.99    58.4 2027.92    61.7  2019.9
    64.9 2010.79    68.2 2006.81   70.62 2006.33    74.7  2006.1    81.2  2006.3
    94.1 2009.72   103.9 2010.81   107.1 2011.95   116.9 2017.04   120.1 2018.08
   123.4  2018.6   126.6 2018.54   133.1 2017.84   149.3 2016.73   155.8 2016.63
   159.1 2017.17     172  2020.6   181.8 2021.69     198 2025.02   217.5 2027.28
#Mann= 3 ,-1 , 0
       0     .12       0   70.62    .045       0    81.2     .12       0
Bank Sta=70.62,81.2
XS Rating Curve= 0 ,0
Exp/Cntr=0.3,0.1

Type RM Length L Ch R = 1 ,9462.5  ,150.5,148.6,146.1
XS GIS Cut Line= 3
     1970811.942      235118.987     1970775.273      235072.317
     1970637.486       235037.87
#Sta/Elev= 30
       0 2066.25     9.4 2061.03    18.7 2055.26    37.5 2044.14    46.9 2038.12
      50 2035.84    53.1 2033.35    56.2 2030.57    59.4 2027.37    65.8 2021.56
    72.3 2014.34    78.7 2006.17      82 2003.66    85.2  2002.7    91.6  2002.4
   101.3 2002.53   107.8 2003.19   114.2 2004.14   117.4 2005.34   123.9 2008.91
   127.1 2009.94   133.6 2010.47   136.8 2011.13   143.3 2013.26   146.5 2013.86
   162.6 2015.08   165.9 2015.13   172.3  2015.1     182 2014.24   201.4 2013.68
#Mann= 3 ,-1 , 0
       0     .12       0    85.2    .045       0   101.3     .12       0
Bank Sta=85.2,101.3
XS Rating Curve= 0 ,0
Exp/Cntr=0.3,0.1

Type RM Length L Ch R = 1 ,9314    ,149,171.8,193.7
XS GIS Cut Line= 2
     1970846.389      234928.974     1970671.933      234903.417
#Sta/Elev= 30
       0 2005.19     9.8 2005.82    19.6 2005.59    32.6 2006.46    39.2 2007.52
    42.4 2007.81    45.7 2007.61      49 2006.55    58.8 2000.95      62 1999.44
    68.6 1997.67   76.28 1996.28    81.6 1995.73    84.9 1995.75    89.5 1996.25
    91.4  1996.5    94.7 1997.57      98 1999.66   101.2 2001.38     111  2002.9
   120.8 2005.61   124.1 2006.29   130.6  2007.1   143.7 2007.14   150.2 2007.88
   153.5 2008.96   156.7 2010.65   166.5  2016.6     173 2019.92   176.3 2021.93
#Mann= 3 ,-1 , 0
       0     .12       0   76.28    .045       0    89.5     .12       0
Bank Sta=76.28,89.5
XS Rating Curve= 0 ,0
Exp/Cntr=0.3,0.1

Type RM Length L Ch R = 1 ,9142.2  ,134.7,154.1,171.1
XS GIS Cut Line= 2
     1970849.722      234854.525     1970770.828      234697.847
#Sta/Elev= 30
       0 2000.59     9.8 1999.03    19.5 1998.28      39 1999.51    45.5 1999.17
      65 1995.25    68.2 1995.05      78 1996.41    84.5 1996.56    87.7 1996.05
      91 1994.17    94.2 1991.61    97.5 1990.55     104 1990.09   113.7 1989.93
     117 1990.03   123.4  1990.7   126.7 1991.65   133.2  1994.6   136.4 1996.94
   139.7 2002.47   142.9 2013.24   146.2 2025.53   149.4  2033.9   152.7 2040.52
   155.9  2045.3   162.4  2053.1   165.7 2056.67   172.2 2062.21   175.4  2065.5
#Mann= 3 ,-1 , 0
       0     .12       0     104    .045       0     117     .12       0
Bank Sta=104,117
XS Rating Curve= 0 ,0
Exp/Cntr=0.3,0.1

Type RM Length L Ch R = 1 ,8988.1  ,160.8,142.2,123
XS GIS Cut Line= 3
     1970908.615      234872.304      1970950.84      234752.295
     1970904.171      234690.069
#Sta/Elev= 30
       0 2001.32     3.3 2000.82     9.8 1998.94    19.6 1998.01    22.8 1997.48
    29.4 1995.37    39.1 1991.62    42.4 1990.53    48.9  1989.1    58.7 1985.71
    65.2 1983.04   67.05 1982.68    71.8  1982.3    78.3 1982.43   79.85 1982.69
    81.6 1982.98    88.1 1985.71    91.3 1986.48   110.9 1988.85   120.7    1991
   130.5 1992.32   136.9 1993.75   140.2 1994.84   146.7 1997.42   156.4 2002.22
   169.4    2008   175.8 2011.29   185.6 2015.85   201.8 2023.95     205 2025.76
#Mann= 3 ,-1 , 0
       0     .12       0   67.05    .045       0   79.85     .12       0
Bank Sta=67.05,79.85
XS Rating Curve= 0 ,0
Exp/Cntr=0.3,0.1

Type RM Length L Ch R = 1 ,8845.8  ,174.2,162.6,150.5
XS GIS Cut Line= 2
      1971109.74      234855.636     1971020.845       234691.18
#Sta/Elev= 30
       0 2040.83     9.8 2033.33      23 2023.78    29.5 2018.64    32.8  2015.6
    39.4 2007.19    42.6 2003.78    45.9 2001.74    52.5 1999.03    55.8 1996.63
      59 1993.29    68.9  1982.3    72.2 1980.08    75.4 1979.09    78.7 1978.63
    85.3 1978.38    91.8 1978.69    95.1 1979.38    98.4 1980.53     105 1982.08
   111.5 1983.93   118.1 1985.12   121.4  1985.1   134.5 1983.88   137.8 1984.18
     141 1985.02   147.6  1987.5     164 1990.47   177.1 1991.06   186.9 1990.79
#Mann= 3 ,-1 , 0
       0     .12       0    78.7    .045       0    91.8     .12       0
Bank Sta=78.7,91.8
XS Rating Curve= 0 ,0
Exp/Cntr=0.3,0.1

Type RM Length L Ch R = 1 ,8683.3  ,153.3,152.8,152
XS GIS Cut Line= 2
     1971267.529       234728.96      1971099.74       234625.62
#Sta/Elev= 30
       0 2029.31     3.2 2028.41     6.5 2026.87     9.7 2024.15    16.2  2016.8
    19.4 2013.95    25.8 2008.79    35.5 2001.58    54.9 1987.39    58.2 1985.26
    64.6 1977.89    67.8 1976.46    77.5 1975.74      84 1975.13    90.4 1975.62
    93.7 1976.28    96.9 1977.64   106.6 1984.18   109.8 1985.34   122.8 1987.22
   135.7  1988.2   142.1 1988.48   158.3 1988.21   164.8 1988.56     168 1988.41
   174.4 1987.59   184.1  1984.4   190.6 1982.91   193.8  1982.5   197.1 1982.46
#Mann= 3 ,-1 , 0
       0     .12       0    77.5    .045       0    90.4     .12       0
Bank Sta=77.5,90.4
XS Rating Curve= 0 ,0
Exp/Cntr=0.3,0.1

Type RM Length L Ch R = 1 ,8530.4  ,167,165.3,163.4
XS GIS Cut Line= 2
     1971355.313      234601.174     1971174.189      234496.722
#Sta/Elev= 30
       0 2016.35     3.3 2016.28     6.5  2015.7    16.3 2011.88    22.9 2009.89
    29.4 2007.51    35.9 2006.14    39.2    2005    42.5 2003.72    45.7 2002.05
    52.3 1997.06    55.5 1994.37    75.1 1977.27    84.9 1969.76    88.2 1968.09
    94.2 1966.72      98 1966.53   107.8 1966.83   111.1 1967.63   114.3 1969.04
   130.7  1977.7   133.9    1979   137.2 1979.65   143.7 1980.01   153.6 1981.61
   160.1 1982.11   169.9 1981.55   179.7 1979.83   199.3 1980.08   209.1 1979.68
#Mann= 3 ,-1 , 0
       0     .12       0    94.2    .045       0   107.8     .12       0
Bank Sta=94.2,107.8
XS Rating Curve= 0 ,0
Exp/Cntr=0.3,0.1

Type RM Length L Ch R = 1 ,8365.1  ,209.7,208.7,207.6
XS GIS Cut Line= 2
     1971433.096      234450.053     1971236.416      234356.713
#Sta/Elev= 30
       0 1995.57     9.8 1995.18      13 1993.91      26 1985.42    35.7 1978.68
    42.2 1975.04    48.7 1972.11    55.2 1970.37    61.7 1967.41    68.2 1965.99
    71.7 1964.91    74.7    1964      78 1963.85    86.7 1965.12    97.5 1967.21
     104 1968.08     117 1968.58     130 1968.42   149.5 1968.87   152.7 1969.37
     156 1970.32   162.5  1972.8   165.7  1973.7     169  1974.2   178.7  1975.2
   188.5 1975.52   198.2 1977.11     208 1978.21   214.5 1978.54   217.7  1978.2
#Mann= 3 ,-1 , 0
       0     .12       0    71.7    .045       0    86.7     .12       0
Bank Sta=71.7,86.7
XS Rating Curve= 0 ,0
Exp/Cntr=0.3,0.1

Type RM Length L Ch R = 1 ,8156.4  ,218.2,209.2,199.5
XS GIS Cut Line= 2
     1971572.381      234278.152     1971276.724      234154.961
#Sta/Elev= 30
       0 2023.34     3.3 2020.29     6.5 2017.84    22.9 2006.95    45.8 1990.72
    78.4  1968.3      85 1963.28    88.2 1961.29    91.5 1960.59   101.3 1960.69
   114.4 1959.91   124.2 1958.02     134 1957.53  139.11 1957.98   156.9 1960.46
   163.4 1959.28   179.8 1957.39   186.3 1958.57   196.1 1962.71   199.4 1963.82
   202.6 1964.31   212.4 1964.59   228.8 1965.67   235.3 1965.52   241.9 1965.97
   254.9 1967.55   271.3 1967.05   287.6 1967.52     304 1969.16   320.3  1971.6
#Mann= 3 ,-1 , 0
       0     .12       0   124.2    .045       0  139.11     .12       0
#XS Ineff= 2 , 0
          110.53 1963.11  157.12         1963.51
Permanent Ineff=
       F       F
Bank Sta=124.2,139.11
XS Rating Curve= 0 ,0
Exp/Cntr=0.3,0.1

Type RM Length L Ch R = 1 ,7947.2  ,177.9,181.5,184.2
XS GIS Cut Line= 2
     1971631.923      234033.824     1971342.425       234037.93
#Sta/Elev= 30
       0 2041.52     9.8 2035.19    22.8 2025.57    32.5 2017.15      39 2011.99
    48.8 2003.35    55.3 1997.15    61.8  1990.2    68.3 1984.25    71.6 1979.77
    81.3 1961.81    87.8 1951.63    91.1 1947.74    94.3 1945.53    97.6 1944.72
   100.8 1944.49   110.6 1944.72   120.4 1945.62   130.1 1947.51   143.1 1948.18
   152.9 1952.73   159.4 1955.12   165.9 1956.72   182.2 1959.46   191.9 1959.41
   211.4 1956.45   214.7 1956.41   247.2 1959.91   276.5 1960.24   289.5 1960.87
#Mann= 3 ,-1 , 0
       0     .12       0    97.6    .045       0   110.6     .12       0
#XS Ineff= 2 , 0
                          130.65         1951.35
Permanent Ineff=
       F       F
Bank Sta=97.6,110.6
XS Rating Curve= 0 ,0
Exp/Cntr=0.3,0.1

Type RM Length L Ch R = 1 ,7765.7  ,208.9,217.4,224.7
XS GIS Cut Line= 2
     1971658.614      233875.729      1971404.02      233844.932
#Sta/Elev= 30
       0 2027.23    19.5 2016.56    51.9 1997.39    55.2 1995.76    61.7 1991.79
    68.2 1986.85    71.4 1983.82    74.7 1979.95    81.2 1973.57    90.9 1961.22
    94.1 1957.03    97.4 1952.15   103.9 1940.73   107.1 1938.29   110.4 1936.66
  115.49 1935.34   116.9 1935.08   129.8 1935.32   139.6 1936.35   152.6 1939.82
   159.1 1941.18     172 1942.36   178.5 1944.25   188.3  1948.4   194.8 1949.44
     211 1948.61   227.2 1948.63     237 1949.05     250 1948.52   256.4 1948.64
#Mann= 3 ,-1 , 0
       0     .12       0  115.49    .045       0   129.8     .12       0
Bank Sta=115.49,129.8
XS Rating Curve= 0 ,0
Exp/Cntr=0.3,0.1

Type RM Length L Ch R = 1 ,7548.3  ,235.4,236.1,235.4
XS GIS Cut Line= 2
     1971664.774      233750.486     1971412.233      233627.295
#Sta/Elev= 30
       0  2007.1     6.5 2002.59    19.6 1994.58    45.7    1977    55.5 1971.37
    81.7 1955.09    88.2 1950.76    94.8 1946.84   107.8 1938.17   114.4 1934.35
   120.9 1931.74   127.4 1930.45     134 1930.24   143.8 1931.25   153.6 1930.79
   156.8 1929.59   160.1 1927.63   163.4 1926.22  174.94 1925.63     183 1924.98
   186.2 1924.98   189.5 1925.69     196 1927.96   209.1 1931.94   218.9 1933.52
   225.4 1934.16   235.2 1936.64   251.6 1938.88   271.2 1939.53     281 1943.97
#Mann= 3 ,-1 , 0
       0     .12       0  174.94    .045       0   189.5     .12       0
Bank Sta=174.94,189.5
XS Rating Curve= 0 ,0
Exp/Cntr=0.3,0.1

Type RM Length L Ch R = 1 ,7312.2  ,256.2,250.5,242.5
XS GIS Cut Line= 3
      1971714.05      233543.115     1971670.933      233495.892
     1971510.785      233417.871
#Sta/Elev= 30
       0 1957.41    22.4    1947      32 1943.22    41.6 1937.96    51.2  1936.3
    57.6 1933.02    67.2 1929.93    76.9 1928.13    89.9 1928.93    93.1 1928.33
    96.3 1926.15     106 1918.45   109.3 1916.97   112.2 1916.36   115.8 1916.04
   125.5 1916.38   135.2 1917.03   144.9  1919.2   148.2  1920.8   151.4 1923.49
   154.6 1925.47   157.9 1926.56   180.6 1927.31   193.5 1927.22     200 1927.74
   203.2 1928.74   212.9 1933.73   216.2 1935.86   229.1 1945.74   242.1 1954.14
#Mann= 3 ,-1 , 0
       0     .12       0   112.2    .045       0   125.5     .12       0
Bank Sta=112.2,125.5
XS Rating Curve= 0 ,0
Exp/Cntr=0.3,0.1

Type RM Length L Ch R = 1 ,7061.7  ,287.4,284.5,281.2
XS GIS Cut Line= 2
     1971818.762       233261.83     1971570.328       233222.82
#Sta/Elev= 30
       0 1928.45     9.8 1927.93    45.7  1924.3    58.8 1922.69    68.6 1921.06
    75.1  1919.4    78.4 1917.98    81.6  1915.8    88.2 1909.99    91.4 1909.63
   101.2 1909.58   104.5 1909.27   114.3 1908.82   120.8 1909.32   130.6 1913.06
   140.4 1913.36     147 1914.65   150.2 1914.83   153.5 1915.56   156.8 1916.88
   173.1 1925.59   176.4    1927   182.9 1930.69   192.7 1937.27   205.8  1944.6
   212.3 1948.75   218.8 1952.47   238.4 1965.58   248.2 1971.36   251.5 1973.84
#Mann= 3 ,-1 , 0
       0     .12       0   104.5    .045       0   120.8     .12       0
Bank Sta=104.5,120.8
XS Rating Curve= 0 ,0
Exp/Cntr=0.3,0.1

Type RM Length L Ch R = 1 ,6777.2  ,310.5,302.5,292.4
XS GIS Cut Line= 3
     1971845.453       232964.12      1971623.71      232960.014
     1971551.849      232984.652
#Sta/Elev= 30
       0 1916.74     6.5 1916.69     9.8  1915.6    16.3 1911.13    19.6 1909.57
    26.1 1908.26    45.7 1907.56    58.7 1906.27    81.5 1907.33    88.1  1906.4
    97.8 1903.42   114.2 1901.82   124.4 1899.42     137 1899.08   140.2 1899.31
   143.5 1900.66     150 1904.64   153.3 1905.52   163.1 1906.77   172.9 1907.23
   189.2 1905.57   202.2 1905.44     225 1907.52   231.3 1910.14   240.8 1916.38
   247.1 1917.76   250.3  1919.2   259.8 1926.84   269.3 1932.27   297.8 1951.02
#Mann= 3 ,-1 , 0
       0     .12       0   124.4    .045       0   140.2     .12       0
Bank Sta=124.4,140.2
XS Rating Curve= 0 ,0
Exp/Cntr=0.3,0.1

Type RM Length L Ch R = 1 ,6474.7  ,211.9,212.2,212.3
XS GIS Cut Line= 2
     1971771.539      232670.516     1971484.094      232781.387
#Sta/Elev= 30
       0 1946.08     3.3 1944.29    13.1 1942.84    22.9 1936.33    39.3 1928.15
    68.8 1917.56    78.7 1916.42    91.8 1910.51    98.3  1907.1   101.6 1903.38
   108.2 1894.26   111.4 1891.24     118 1888.32   127.8 1887.61   137.7 1887.15
  144.61 1887.63   157.3 1895.19   160.6 1896.74   167.2 1898.36   183.5 1898.78
   199.9 1898.01   219.6 1899.63   239.3 1898.67   255.6 1901.54   262.2  1904.3
   278.6 1914.44   285.1 1919.46     295 1925.82   301.5 1931.95   308.1 1936.79
#Mann= 3 ,-1 , 0
       0     .12       0   127.8    .045       0  144.61     .12       0
Bank Sta=127.8,144.61
XS Rating Curve= 0 ,0
Exp/Cntr=0.3,0.1

Type RM Length L Ch R = 1 ,6262.5  ,215.7,230,244.4
XS GIS Cut Line= 2
     1971672.986      232483.677     1971420.446      232580.176
#Sta/Elev= 30
       0 1928.34     6.5  1925.4      13 1921.56    16.3 1920.45    26.1 1919.27
    39.1 1913.93    52.1 1911.44    65.1 1906.39    71.7 1905.23    78.2 1904.96
    94.5 1900.79     101 1898.46   104.2 1897.03   107.5  1894.8   120.5 1883.99
   123.8 1881.92  125.81 1881.29   130.3  1880.6   140.1 1881.25   153.1 1883.39
   159.6 1883.91   185.7 1892.08   188.9 1892.74   211.7 1893.22   221.5 1892.59
     228 1892.69   247.6  1898.9   250.8 1900.42   260.6 1906.82   270.4 1914.59
#Mann= 3 ,-1 , 0
       0     .12       0  125.81    .045       0   140.1     .12       0
Bank Sta=125.81,140.1
XS Rating Curve= 0 ,0
Exp/Cntr=0.3,0.1

Type RM Length L Ch R = 1 ,6032.5  ,231.2,214.1,196.4
XS GIS Cut Line= 3
     1971648.348      232376.912     1971414.286      232313.264
     1971305.468       232362.54
#Sta/Elev= 30
       0 1924.93    42.6 1911.44    52.4  1907.5    62.3 1901.94    78.7 1891.55
      82 1889.84    85.2 1888.83    95.1 1887.64   101.6 1886.25   131.1 1882.08
   147.5 1880.83   150.8    1880   157.3 1876.69   163.9  1874.3   170.4 1872.79
   173.7 1872.62   183.6  1872.8   190.1 1872.81   193.4 1873.26   203.2 1876.37
   206.5  1876.8   222.9 1876.49   229.4 1877.36     236 1878.82   242.6 1882.09
   255.5 1890.09   274.8 1903.98     291 1913.94   300.7 1921.27     362 1964.35
#Mann= 3 ,-1 , 0
       0     .12       0   170.4    .045       0   183.6     .12       0
Bank Sta=170.4,183.6
XS Rating Curve= 0 ,0
Exp/Cntr=0.3,0.1

Type RM Length L Ch R = 1 ,5818.4  ,258.8,243.1,226.2
XS GIS Cut Line= 2
     1971592.912      232085.361     1971272.617      232257.828
#Sta/Elev= 30
       0 1960.87     9.8 1952.34    19.7 1942.63    29.5 1933.91      36  1926.9
    42.6 1916.61    52.4 1899.86    65.6 1882.94    81.9 1870.24   91.17 1866.23
      95 1865.53   104.9 1866.25   111.4  1866.9   134.4  1873.5   140.9  1874.7
   157.3 1875.15   170.4 1874.04   183.5 1874.32   186.8 1874.87   199.9 1878.91
   226.1 1878.25     236 1878.76   242.5 1879.89   255.6  1885.1   285.1 1900.82
   291.7  1903.3   304.8 1911.74   340.8 1932.64   357.2 1943.55   363.8 1946.72
#Mann= 3 ,-1 , 0
       0     .12       0   91.17    .045       0   104.9     .12       0
Bank Sta=91.17,104.9
XS Rating Curve= 0 ,0
Exp/Cntr=0.3,0.1

Type RM Length L Ch R = 1 ,5575.3  ,302.6,321.4,339.4
XS GIS Cut Line= 4
     1971414.286       231884.15     1971332.159      231935.479
     1971278.777      232077.148     1971188.437      232146.956
#Sta/Elev= 30
       0 1909.04    22.6 1893.57      42 1882.42    58.1 1876.39    64.6 1874.76
    74.2 1874.06    96.8 1871.38   122.6  1870.6   132.3 1867.73   135.5 1866.14
   138.7 1863.83   141.9 1860.71   145.2 1858.62   149.2 1857.39     158 1856.42
   164.2 1857.39   177.4 1860.75   180.6 1861.14   203.2 1860.35   206.4  1860.5
   209.6 1861.28   212.8 1862.78     216 1864.95   232.1 1878.51   241.8 1884.57
     258 1892.64   277.6 1901.67   313.5    1917   349.4 1934.75   362.4 1942.31
#Mann= 3 ,-1 , 0
       0     .12       0   149.2    .045       0   164.2     .12       0
Bank Sta=149.2,164.2
XS Rating Curve= 0 ,0
Exp/Cntr=0.3,0.1

Type RM Length L Ch R = 1 ,5253.8  ,316.3,323.5,329.7
XS GIS Cut Line= 3
     1971295.202      231719.896     1971089.885      231804.076
     1971050.874       231974.49
#Sta/Elev= 30
       0 1899.33    16.3 1891.58    35.9 1883.37    55.5 1874.29    65.3 1871.68
    75.1 1867.65    84.8 1865.58    91.4 1863.65   101.2 1862.87   104.4  1861.2
     111 1851.23  112.93 1850.14   114.2 1849.42   117.5 1849.17   130.5 1850.15
   133.8 1850.94   143.6 1852.04     173 1853.02     186 1853.89   202.3 1856.09
   218.6 1857.38   225.1 1858.65   238.1  1863.8   257.5  1873.5   276.9 1881.87
   315.8 1895.57   341.7 1900.79   361.1 1906.44   374.1 1911.44   396.7 1921.42
#Mann= 3 ,-1 , 0
       0     .12       0  112.93    .045       0   130.5     .12       0
Bank Sta=112.93,130.5
XS Rating Curve= 0 ,0
Exp/Cntr=0.3,0.1

Type RM Length L Ch R = 1 ,4930.3  ,386.4,396.5,401.8
XS GIS Cut Line= 2
     1971165.852      231537.164     1970747.005      231592.599
#Sta/Elev= 30
       0 1887.26      36 1869.57    45.8 1866.36    52.4 1863.19      59 1862.35
    88.4 1851.57   140.8 1846.75   180.1 1844.94     190  1843.5   193.2 1842.38
   196.5 1842.19   209.6 1843.81     222 1841.45   229.3 1840.87     237 1841.53
   252.2  1840.5   255.5 1840.73   258.7 1844.66   265.3 1854.75   268.6 1857.54
   278.4 1863.77   284.9 1870.35   294.8 1877.45   311.1 1892.51   327.5 1900.28
   347.2 1907.45   363.6  1911.6   373.4 1916.24     393  1928.7   422.5 1950.46
#Mann= 3 ,-1 , 0
       0     .12       0     222    .045       0     237     .12       0
#XS Ineff= 2 , 0
          208.98 1846.28
Permanent Ineff=
       F       F
Bank Sta=222,237
XS Rating Curve= 0 ,0
Exp/Cntr=0.3,0.1

Type RM Length L Ch R = 1 ,4533.8  ,233,231.2,229.5
XS GIS Cut Line= 3
     1971216.365      231229.491     1970963.486      231187.996
     1970861.982      231186.071
#Sta/Elev= 30
       0 1920.53      26 1905.75    42.2 1895.69    58.4 1884.66    77.8 1874.71
    84.3 1871.95    97.3 1862.23     107 1856.88     120 1846.77   142.7 1831.86
   149.2 1828.56   155.7 1827.77   165.4 1827.54   171.9 1827.71   175.2 1828.42
   188.1  1833.1   207.6 1837.16     240 1838.39   243.3 1839.46   256.3 1846.55
   279.2 1861.13   298.8 1876.55   305.4  1880.5   308.7 1883.72   318.5 1898.77
   321.8 1902.61   331.6 1911.92   338.1 1917.23   351.2 1929.18   357.8 1934.01
#Mann= 3 ,-1 , 0
       0     .12       0   155.7    .045       0   171.9     .12       0
Bank Sta=155.7,171.9
XS Rating Curve= 0 ,0
Exp/Cntr=0.3,0.1

Type RM Length L Ch R = 1 ,4302.6  ,293.2,285.8,278
XS GIS Cut Line= 2
     1971204.862       230984.86     1970927.684      230962.275
#Sta/Elev= 30
       0  1910.6     9.8 1903.44    32.7 1882.45    62.2 1860.45    78.5 1847.53
    85.1 1841.74    91.6 1835.11    94.9 1828.08    98.2 1822.25   101.4  1820.1
   104.7 1819.69     108 1819.81   114.5 1821.69   117.8 1821.81   130.9 1819.98
     144 1819.64  148.33 1820.02     157 1823.22   160.3 1823.55   166.9 1823.58
   176.7 1821.82     180 1821.98     193  1827.5   199.6 1828.72     229  1829.8
   238.8 1831.25   248.6 1833.87   255.2 1836.34     265 1841.26   278.1 1849.65
#Mann= 3 ,-1 , 0
       0     .12       0   130.9    .045       0  148.33     .12       0
#XS Ineff= 2 , 0
          115.79 1826.35  163.16         1827.36
Permanent Ineff=
       F       F
Bank Sta=130.9,148.33
XS Rating Curve= 0 ,0
Exp/Cntr=0.3,0.1

Type RM Length L Ch R = 1 ,4016.8  ,219.2,227.8,233.5
XS GIS Cut Line= 3
      1971196.65      230717.947     1971059.087      230687.149
     1970911.258       230726.16
#Sta/Elev= 30
       0 1924.43     9.8 1918.58    29.5 1906.02    45.9  1894.9    55.7 1889.54
    72.1 1879.72    88.5 1870.71   101.6 1864.15   111.5 1858.42   114.7  1855.9
   121.3 1850.06   124.6 1846.78     141  1824.9   147.5  1815.4   150.7 1811.69
  152.08 1811.16     154 1810.42   157.2 1810.13   160.5 1810.15     167 1811.29
   170.1 1812.04   176.8 1813.02   183.3 1813.16   186.5 1813.52     193 1815.62
   212.5 1816.66   241.8 1819.02   251.6 1820.15   271.1 1824.05   293.9 1826.46
#Mann= 3 ,-1 , 0
       0     .12       0  152.08    .045       0     167     .12       0
Bank Sta=152.08,167
XS Rating Curve= 0 ,0
Exp/Cntr=0.3,0.1

Type RM Length L Ch R = 1 ,3789    ,199.5,217.7,235.1
XS GIS Cut Line= 3
      1971196.65      230580.384     1971040.608      230483.885
     1970857.876      230481.832
#Sta/Elev= 30
       0  1904.3     9.8 1899.19    19.7 1894.66    42.6 1885.84    49.1 1883.83
    52.4 1883.15    75.4 1876.81   104.8 1870.42   111.4 1867.96   114.7 1866.22
   117.9 1864.13   124.5 1859.18   147.4 1840.28   157.3 1832.55   186.7 1812.41
     190 1810.82   196.5 1808.76   216.1 1807.86   222.6 1807.89   235.7 1807.34
     239 1807.83     252 1811.53     265  1812.7   271.6 1815.07   281.4 1814.29
   304.2 1815.37   317.3 1816.95   333.6  1819.5   356.4 1821.02   366.2 1822.02
#Mann= 3 ,-1 , 0
       0     .12       0   222.6    .045       0     239     .12       0
Bank Sta=222.6,239
XS Rating Curve= 0 ,0
Exp/Cntr=0.3,0.1
